--- FISHHAWKCK.prj (project) ---

Proj Title=FISHHAWKCK
Current Plan=p01
Default Exp/Contr=0,0
English Units
Geom File=g01
Flow File=f01
Plan File=p01
Background Map Layer=Inundation Boundary (P100yr Value_0)
BEGIN DESCRIPTION:
----------MODEL BY WOOD PLC 2022----------
AFH study
Randolph County, WV
HEC-RAS Version: RAS 6.2
Vertical Datum: NAVD88
Projection: NAD 1983 StatePlane West Virginia S FIPS 4702 (US Feet)
Terrain: 1-meter LIDAR (FEMA Region III 3DEP collected 2016-2018)
Land Use: 2019 NLCD
Hydrologic Method:
WV SIR2010-5033 regression equations
Additional Model Notes:
None
END DESCRIPTION:
DSS Export Rating Curves= 0
DSS Export Rating Curve Sorted= 0
DSS Export Volume Flow Curves= 0
DXF OffsetX= 0
DXF OffsetY= 0
DXF ScaleX= 0
DXF ScaleY= 0

--- FISHHAWKCK.p01 (plan) ---

Plan Title=Floodplain
Program Version=6.20
Short Identifier=Floodplain
Geom File=g01
Flow File=f01
Subcritical Flow
K Sum by GR= 0
Std Step Tol= 0.01
Critical Tol= 0.01
Num of Std Step Trials= 20
Max Error Tol= 0.3
Flow Tol Ratio= 0.001
Split Flow NTrial= 30
Split Flow Tol= 0.02
Split Flow Ratio= 0.02
Log Output Level= 0
Friction Slope Method= 1
Unsteady Friction Slope Method= 2
Unsteady Bridges Friction Slope Method= 1
Parabolic Critical Depth
Global Vel Dist= 0 , 0 , 0
Global Log Level= 0
CheckData=False
Encroach Param=-1 ,0,0, 0
Mapping Interval=1HOUR
Computation Time Step Use Courant=        0
Computation Time Step Use Time Series=    0
Computation Time Step Count To Double=0
Computation Time Step Max Doubling=0
Computation Time Step Max Halving=0
Computation Time Step Residence Courant=0
Run HTab= 0
Run UNet= 0
Run Sediment= 0
Run PostProcess= 0
Run WQNet= 0
Run RASMapper=-1
UNET Theta= 0
UNET Theta Warmup= 0
UNET ZTol= 0
UNET ZSATol= 0
UNET MxIter= 0
UNET Max Iter WO Improvement= 0
UNET MaxInSteps= 0
UNET DtIC= 0
UNET DtMin= 0
UNET MaxCRTS= 0
UNET WFStab= 0
UNET SFStab= 0
UNET WFX= 1
UNET SFX= 1
UNET Gravity=32.174
UNET 1D Methodology=Finite Difference
UNET DSS MLevel= 1
UNET Pardiso=0
UNET DZMax Abort= 0
UNET Use Existing IB Tables= 0
UNET Froude Reduction=False
UNET Froude Limit= 0
UNET Froude Power= 0
UNET D1 Cores= 0
UNET WindReference=Eulerian
UNET WindDragFormulation=Hsu (1988)
UNET D2 Coriolis=0
UNET D2 Cores= 0
UNET D2 Theta= 1
UNET D2 Theta Warmup= 1
UNET D2 Z Tol= 0.01
UNET D2 Volume Tol= 0.01
UNET D2 Max Iterations= 20
UNET D2 Equation= 0
UNET D2 RampUpFraction=0.1
UNET D2 TimeSlices= 1
UNET D2 Turbulence Formulation=Non-Conservative (original)
UNET D2 Eddy Viscosity=0.3
UNET D2 Transverse Eddy Viscosity=0.1
UNET D2 Smagorinsky Mixing=0
UNET D2 BCVolumeCheck=0
UNET D2 Cores=0
UNET D2 SolverType=PARDISO (Direct)
UNET D2 Minimum Iterations= 2147483647
UNET D2 Maximum Iterations= 2147483647
UNET D2 Restart Number= 10
UNET D2 Relaxation Coeff=1.3
UNET D2 SOR Precondition Iterations= 10
UNET D2 ILUT Maximum Fill= 8
UNET D2 ILUT Tolerance=1E-08
UNET D1D2 MaxIter= 0
UNET D1D2 ZTol=0.01
UNET D1D2 QTol=0.1
UNET D1D2 MinQTol=1
Write IC File= 0
Write IC File at Fixed DateTime=0
Write IC File at Sim End=0
Echo Input=False
Echo Parameters=False
Echo Output=False
Write Detailed= 0
HDF Write Warmup=0
HDF Write Time Slices=0
HDF Flush=0
HDF Compression= 1
HDF Chunk Size= 1
HDF Spatial Parts= 1
HDF Use Max Rows=0
HDF Fixed Rows= 1
Calibration Method= 0
Calibration Iterations= 20
Calibration Max Change=0.05
Calibration Tolerance=0.2
Calibration Maximum=1.5
Calibration Minimum=0.5
Calibration Optimization Method= 1
WQ AD Non Conservative
WQ ULTIMATE=-1
WQ Max Comp Step=1HOUR
WQ Output Interval=15MIN
WQ Output Selected Increments= 0
WQ Output face flow=0
WQ Output face velocity=0
WQ Output face area=0
WQ Output face dispersion=0
WQ Output cell volume=0
WQ Output cell surface area=0
WQ Output cell continuity=0
WQ Output cumulative cell continuity=0
WQ Output face conc=0
WQ Output face dconc_dx=0
WQ Output face courant=0
WQ Output face peclet=0
WQ Output face adv mass=0
WQ Output face disp mass=0
WQ Output cell mass=0
WQ Output cell source sink temp=0
WQ Output nsm pathways=0
WQ Output nsm derived pathways=0
WQ Create Restart=0
WQ Fixed Restart=0
WQ System Summary=0
WQ Write To DSS=0
Sorting and Armoring Iterations= 10
XS Update Threshold= 0.02
Bed Roughness Predictor= 0
Hydraulics Update Threshold= 0.02
Energy Slope Method= 1
Volume Change Method= 1
Sediment Retention Method= 0
Sediment TS Multiplier= 1
Warm Up Method= 0
XS Weighting Method= 0
Number of US Weighted Cross Sections= 1
Number of DS Weighted Cross Sections= 1
Upstream XS Weight=0
Main XS Weight=1
Downstream XS Weight=0
Number of DS XS's Weighted with US Boundary= 1
Upstream Boundary Weight= 1
Weight of XSs Associated with US Boundary= 0
Number of US XS's Weighted with DS Boundary= 1
Downstream Boundary Weight= 0.5
Weight of XSs Associated with DS Boundary= 0.5
Percentile Method= 0
Sediment Output Level= 3
Mass or Volume Output= 0
Output Increment Type= 1
Profile and TS Output Increment= 1
Transport Output Increment 1
XS Output Flag= 0
XS Output Increment= 10
Read HDF5 Sediment Hotstart= 0
Sediment Hotstart Type= 0
Write Gradation File= 0
Read Gradation Hotstart= 0
Write HDF5 File= 1
Write Binary Output= 1
Write DSS Sediment File= 0
DSS Sediment Output Type= 1
SV Curve= 0
Specific Gage Flag= 0
Subcell Erosion Methods= 0
Subcell Deposition Methods= 0
Advection Scheme= 1
Matrix Solver= 0
Implicit Weighting Factor= 1
Maximum Outer Loop Convergence Iterations= 5
Convergence Maximum Absolute= 0.001
Convergence RMSE= 0.0001
Grain Fractions Max Abs Error= 0.001
Max Subgrid Regions= 1
Max Subgrid Length Scale= 3.402823E+38
Initial Layer Thickness= 3.402823E+38
Min Layer Thickness= 3.402823E+38
Max Layer Thickness= 3.402823E+38
Number of Layers= 5

--- FISHHAWKCK.f01 (steady flow) ---

Flow Title=Flow
Program Version=6.20
Number of Profiles= 1
Profile Names=P100yr
River Rch & RM=FISHHAWKCK,Main,15521
     472
River Rch & RM=FISHHAWKCK,Main,10862
     531
River Rch & RM=FISHHAWKCK,Main,7608
     668
River Rch & RM=FISHHAWKCK,Main,5204
    1080
Boundary for River Rch & Prof#=FISHHAWKCK,Main            , 1
Up Type= 0
Dn Type= 3
Dn Slope=0.078
DSS Import GetInterval= 0
DSS Import GetPeak= 0
DSS Import FillOption= 0

--- FISHHAWKCK.g01 (geometry) ---

Geom Title=Geometry
Program Version=6.20

River Reach=FISHHAWKCK      ,Main
Reach XY= 30
2318030.77700001660131.5370000152318337.54700002660319.819000006
2318751.08900002660169.819000006     2318763.589659836.225000009
     2319040.412659783.3599999992320072.38429209658734.159299413
2320591.22199999658819.3320000172320826.89900005658677.665999994
2321042.52399999658781.3120000212321269.86800005659134.175999999
2321296.43000001659716.9889999932321467.48100002659896.306999996
2321287.79300001660206.4630000142321427.59254239660754.047605222
2321350.32693101661023.6366883012321697.38813395661411.490216785
2321654.74300002662047.8390000162322073.45799999662494.488000005
2322471.12395172662538.2271052732322634.96500002662807.512000009
2323570.79128829662838.0151351632323910.27000003662509.343999997
2324275.09900002      662542.8092325090.76000001 662087.36300002
2325456.36000003662194.840000004     2326055.184662093.408000007
2326902.02100001662443.2720000152327250.00100003662868.776999995
     2327334.574 663167.424000012327522.84696178663267.935375451

Type RM Length L Ch R = 1 ,15521   ,395,392.7,384.6
XS GIS Cut Line= 4
2317848.41471146660317.7764745742317991.45758544660222.861399511
2318071.12335832660102.349281501 2318046.6791063659956.661539449
#Sta/Elev= 30
       0    3533    28.5 3522.78    42.9 3518.62    75.3 3514.16   104.1 3512.94
   131.3 3513.26   143.7 3511.35   179.2 3510.55   184.9 3509.98   192.9 3507.43
   197.7 3506.81   231.2 3508.38     236 3507.39   245.6 3503.77   262.9 3501.85
   268.7  3501.2   271.83501.826     286 3505.79   297.5 3508.44   312.7 3508.08
   325.4 3510.79   341.7 3510.94   361.9  3513.8   390.3 3515.25   398.4 3514.82
   402.5 3515.09   426.1 3519.71   434.9 3521.93     439 3522.19   463.9 3526.53
#Mann= 7 ,-1,0
       0      .1       0      20     .12       0   262.9    .045       0
   271.8     .12       0  301.67      .1       0  376.13     .12       0
  386.13      .1       0
Bank Sta=262.9,271.8
XS Rating Curve= 0 ,0
Exp/Cntr(USF)=0,0
Exp/Cntr=0.3,0.1

Type RM Length L Ch R = 1 ,15128   ,176.8,176.2,174.7
XS GIS Cut Line= 4
2318487.62212414660466.5901475752318398.12682864660346.207095216
 2318307.0475456660151.3766288982318220.72022516659867.050867075
#Sta/Elev= 30
       0 3536.28      12    3532    76.5 3517.35   111.4 3507.05   126.4 3504.33
   136.3 3504.98   146.6 3502.61   155.6 3499.62   173.2 3491.36   192.63486.312
   199.7 3485.81   202.63486.325   211.3 3488.43   230.2 3488.08   239.6 3490.08
   251.5 3491.01   274.8 3490.23   287.6 3491.75   320.7 3492.81   344.8 3497.17
   358.7 3503.84   372.3 3505.45   400.8 3505.53   459.3 3503.34   480.2 3505.23
     522 3506.12   574.2 3508.63     609 3515.47   651.3 3525.59   662.2 3526.11
#Mann= 5 ,-1,0
       0      .1       0      60     .12       0   192.6    .045       0
   202.6     .12       0  575.07      .1       0
Bank Sta=192.6,202.6
XS Rating Curve= 0 ,0
Exp/Cntr(USF)=0,0
Exp/Cntr=0.3,0.1

Type RM Length L Ch R = 1 ,14952   ,263.8,266.1,264.1
XS GIS Cut Line= 2
2318647.60486478660372.3428894782318241.31206306659824.283203737
#Sta/Elev= 30
       0 3543.84    53.7  3530.6    98.5 3516.89   113.4 3509.82   153.4  3487.1
   164.8 3485.09   193.8 3484.78   204.9 3482.46   213.1 3481.99   219.2 3482.52
     238 3487.18   267.8 3486.76   287.8 3488.24   302.7 3487.64   327.6 3494.96
   367.4 3498.56   433.6 3500.45   529.7 3499.74   543.1 3501.19   556.6 3499.75
     570  3503.3   581.5  3502.4   591.5  3503.6   596.5 3505.13   606.4 3510.42
   619.5 3514.73   646.3 3517.63   657.3 3520.81     671 3523.25   682.2  3527.8
#Mann= 7 ,-1,0
       0      .1       0      40     .12       0     160      .1       0
     170     .12       0   204.9    .045       0   219.2     .12       0
     660      .1       0
#XS Ineff= 2 , 0
          173.41 3491.95
Permanent Ineff=
       F       F
Bank Sta=204.9,219.2
XS Rating Curve= 0 ,0
Exp/Cntr(USF)=0,0
Exp/Cntr=0.3,0.1

Type RM Length L Ch R = 1 ,14685   ,296,294.7,291.4
XS GIS Cut Line= 2
2318847.18729369660217.1121114362318249.23200072659817.947253613
#Sta/Elev= 30
       0 3540.51    18.1 3535.55    42.5 3522.32    74.2 3499.96    80.6  3494.6
      95 3479.58   100.2 3476.05   104.6 3475.15   108.8  3476.1   114.2  3478.1
     144  3479.1   158.4 3481.55   209.8 3482.88   239.3 3488.79   290.5 3486.19
   336.7 3486.72   360.1 3490.02   382.8  3488.7   397.2 3491.44   411.7 3491.53
   426.8 3494.29   450.9 3494.06   501.1 3496.67   575.9 3496.69     602 3498.27
   619.5 3499.76   639.5 3504.71   669.9 3508.76   691.4 3515.05   718.9 3526.41
#Mann= 5 ,-1,0
       0      .1       0   100.2    .045       0   108.8      .1       0
     120     .12       0     710      .1       0
#XS Ineff= 2 , 0
                          145.72            3486
Permanent Ineff=
       F       F
Bank Sta=100.2,108.8
XS Rating Curve= 0 ,0
Exp/Cntr(USF)=0,0
Exp/Cntr=0.3,0.1

Type RM Length L Ch R = 1 ,14391   ,243.4,254.1,257.4
XS GIS Cut Line= 4
2318928.46932051660030.3775813872318813.19022798659874.618807501
2318703.19109388659869.3388490642318498.15270791659632.620712481
#Sta/Elev= 30
       0 3518.37   115.9 3494.77   141.7 3491.05   170.7 3488.92   206.8 3472.77
   218.8 3470.33   238.2 3470.75     242  3469.3   246.9 3468.47   250.63469.323
   266.9 3474.14   290.9 3474.39   294.3 3475.03   298.9 3476.67   303.9 3479.58
     309 3481.12   317.5 3480.75   326.8 3478.95   331.7 3479.99   339.1 3483.52
   346.5 3485.83   375.7 3489.16     447 3488.77   521.1  3490.5   538.7 3494.41
   546.8 3497.33   555.7 3497.78   575.5 3501.82   595.2  3508.5   617.1 3519.51
#Mann= 5 ,-1,0
       0      .1       0     140     .12       0     242    .045       0
   250.6     .12       0   543.9      .1       0
Bank Sta=242,250.6
XS Rating Curve= 0 ,0
Exp/Cntr(USF)=0,0
Exp/Cntr=0.3,0.1

Type RM Length L Ch R = 1 ,14137   ,306.5,300.8,294.3
XS GIS Cut Line= 4
2319056.06831607659944.1382602532318976.86893952659831.499146934
2318970.70898801659770.779624911 2318773.5905397 659500.62175156
#Sta/Elev= 30
       0 3511.57    13.5 3507.27    28.1 3503.54    52.5 3498.65    65.2 3494.53
      77 3491.75   106.3 3487.54   130.8 3481.49   139.5 3476.64   152.9 3466.56
   164.2 3458.85     1673457.566   176.2 3456.78   182.53457.583   192.3 3460.93
     216 3462.06   235.4 3468.26   245.3 3467.99   267.5 3476.99   273.3 3478.37
   339.1 3479.02   359.1 3478.31   383.9 3478.55   403.7 3479.36   416.4 3481.29
   433.6 3482.53   458.2 3487.03   474.5 3491.13     522 3504.68   533.2 3509.02
#Mann= 5 ,-1,0
       0      .1       0     167    .045       0   182.5      .1       0
  218.73     .12       0  408.73      .1       0
Bank Sta=167,182.5
XS Rating Curve= 0 ,0
Exp/Cntr(USF)=0,0
Exp/Cntr=0.3,0.1

Type RM Length L Ch R = 1 ,13836   ,61.2,61,61
XS GIS Cut Line= 3
2319234.70690985659762.8596872552319180.14733933659621.180802534
2318905.58950062 659418.78239579
#Sta/Elev= 30
       0 3497.07    23.2 3490.63    34.2 3488.57    43.5 3485.42    53.2 3483.66
    62.7  3479.9    83.2 3474.86    96.1 3470.41     109 3469.19     139 3460.85
   148.7 3456.99   166.1 3446.62   176.6 3443.04   183.3 3442.49   191.5 3443.07
     199  3445.7   211.9  3447.2   221.4 3451.81   232.7 3455.83   246.2 3458.72
   266.4 3461.36   283.4 3462.15   295.9 3464.43     332 3466.02   387.8 3474.05
   410.2 3478.91     440  3486.8   464.9 3491.44   474.8 3495.82   492.9  3501.9
#Mann= 4 ,-1,0
       0      .1       0   176.6    .045       0   191.5      .1       0
  201.82     .12       0
Bank Sta=176.6,191.5
XS Rating Curve= 0 ,0
Exp/Cntr(USF)=0,0
Exp/Cntr=0.3,0.1

Type RM Length L Ch R = 1 ,13775   ,72.4,78.8,81.4
XS GIS Cut Line= 3
2319264.62667432659718.8600336152319211.82708996659568.381218166
2318949.58915426659380.942693659
#Sta/Elev= 30
       0 3489.24    17.4 3485.81    27.2  3481.2    78.1 3466.78      99 3462.15
   122.2 3458.26   133.2 3453.69   154.4 3442.19   159.5 3440.89   168.9 3440.78
   181.6 3437.59   184.5 3437.27   190.2 3437.62   199.4  3438.8   232.8 3450.76
   247.5 3452.87   257.4 3455.47   267.2 3456.45   282.1 3456.17   291.8 3457.48
   306.5 3461.69     336 3462.21     345 3464.21   355.7 3465.37   371.3 3469.93
     400 3475.33   414.7 3479.91   445.4 3487.61   460.8 3492.26   481.8 3500.27
#Mann= 6 ,-1,0
       0      .1       0  179.47     .12       0   181.6    .045       0
   190.2     .12       0  349.47      .1       0  369.47     .12       0
Bank Sta=181.6,190.2
XS Rating Curve= 0 ,0
Exp/Cntr(USF)=0,0
Exp/Cntr=0.3,0.1

Type RM Length L Ch R = 1 ,13696   ,229.6,224.7,220.2
XS GIS Cut Line= 4
2319302.46637645659700.3801790862319262.86668818659563.101259729
2319239.98686829659425.8223403722318975.10895337 659362.46283913
#Sta/Elev= 30
       0 3488.66     7.5 3486.42    15.8 3486.21    28.3 3481.31    61.6 3471.87
    91.7 3465.09   103.2 3463.43   111.1 3460.93   128.2 3452.58   136.6 3446.77
   153.8 3433.17   173.2 3426.83   180.2 3425.61   185.1 3425.35   195.5 3425.61
   201.6 3426.35   213.8 3433.75     230 3434.14   246.2 3437.16   254.3 3436.61
     282 3440.09   298.3  3444.1   347.7 3448.55   376.5 3454.02     389  3457.6
   421.7 3461.72   479.3 3473.41   495.7  3478.6   508.1 3481.26   554.4  3498.9
#Mann= 7 ,-1,0
       0      .1       0   180.2    .045       0   195.5      .1       0
  282.05     .12       0  392.05      .1       0  492.05     .12       0
  552.05      .1       0
Bank Sta=180.2,195.5
XS Rating Curve= 0 ,0
Exp/Cntr(USF)=0,0
Exp/Cntr=0.3,0.1

Type RM Length L Ch R = 1 ,13471   ,113.7,113.6,110.8
XS GIS Cut Line= 3
2319571.74425673659536.7014675452319233.82691678659234.863843574
2319073.66817753659232.223864355
#Sta/Elev= 30
       0 3483.34    15.5 3479.39    33.4 3477.35    67.3 3469.49      90 3462.34
    98.5 3461.12   117.4 3454.26   131.4 3451.36   171.1 3434.97   197.4 3418.81
   220.3  3411.2   223.2 3410.63   228.5 3411.19   245.5 3417.38   257.5 3418.02
   271.3 3423.32   287.5 3426.09   317.5 3423.76     345 3428.27   383.6 3429.76
   396.3 3432.75   425.6 3436.04   466.7 3445.19     480 3446.75   510.8 3453.46
   526.8 3458.95   558.8 3466.97     567 3470.91   594.8 3479.17   613.3 3488.16
#Mann= 5 ,-1,0
       0      .1       0     180     .12       0   220.3    .045       0
   228.5     .12       0     450      .1       0
Bank Sta=220.3,228.5
XS Rating Curve= 0 ,0
Exp/Cntr(USF)=0,0
Exp/Cntr=0.3,0.1

Type RM Length L Ch R = 1 ,13358   ,43.1,44,43.6
XS GIS Cut Line= 6
2319606.06398657659503.2617307792319534.78454767659350.142936111
2319468.78506721659299.9833309612319393.10566295659314.063220126
2319250.54678516659193.5041691522319119.42781731659194.384162225
#Sta/Elev= 30
       0  3480.5    24.4 3475.12    64.1 3462.63    90.5 3457.87   152.3 3441.53
   168.9  3434.8   177.2 3430.71   194.3 3419.01   211.4 3404.97   216.13403.016
   228.5 3402.54   234.2 3402.97   256.5 3410.29   280.9 3413.95   313.4 3416.47
   317.5 3417.38   325.6 3421.29   330.1 3421.45   342.5    3419   371.9 3421.06
   382.4 3420.61   398.3 3424.49   423.1 3425.16   477.7 3432.15   534.3  3449.2
   553.8 3450.89   569.8 3454.56   585.8 3456.72   609.8 3464.02   646.6 3473.59
#Mann= 7 ,-1,0
       0      .1       0     160     .12       0   168.9      .1       0
   216.1    .045       0   234.2      .1       0  291.79     .12       0
  525.47      .1       0
Bank Sta=216.1,234.2
XS Rating Curve= 0 ,0
Exp/Cntr(USF)=0,0
Exp/Cntr=0.3,0.1

Type RM Length L Ch R = 1 ,13314   ,66.6,61.7,60.4
XS GIS Cut Line= 6
2319626.74382378659465.4220286482319555.46438488 659312.30323398
2319489.46490442659262.1436288312319413.78550016659276.223517996
2319271.22662237659155.6644670222319140.10765452659156.544460095
#Sta/Elev= 30
       0 3474.71    34.5 3462.95    84.1 3452.04   110.6 3448.11   149.6  3436.4
   163.5 3429.36   173.5 3422.82   193.9 3404.96   203.2  3395.2   207.1 3392.59
   210.1 3392.02   218.2 3391.79   223.3 3392.01   262.4 3398.47   273.4 3404.78
   297.9 3411.77   310.1 3411.19   333.5 3414.55   372.8 3416.01   389.2 3417.77
   401.6 3420.38   432.6 3422.92   467.1 3427.94   482.5 3432.53   493.9 3434.31
   522.5 3443.14   551.8  3448.9   582.5 3458.49   625.8 3465.27   646.6 3472.21
#Mann= 7 ,-1,0
       0      .1       0     120     .12       0   198.9      .1       0
   210.1    .045       0   223.3      .1       0  311.79     .12       0
  508.77      .1       0
Bank Sta=210.1,223.3
XS Rating Curve= 0 ,0
Exp/Cntr(USF)=0,0
Exp/Cntr=0.3,0.1

Type RM Length L Ch R = 1 ,13252   ,37,38.6,40.5
XS GIS Cut Line= 6
2319640.13171273659386.1347480772319568.07992596 659234.03672922
2319465.53840223659209.8112797962319418.72946451659214.335839645
2319276.17058672659093.7767886712319145.05161887659094.656781744
#Sta/Elev= 30
       0 3455.05      32 3449.05    58.6 3442.21    75.8 3439.44    84.8 3436.38
   121.4 3427.93     140 3420.55   151.5 3413.39   160.4 3405.45   168.3 3400.37
   176.4 3392.89   185.6 3389.54     197 3392.57   220.8 3390.47   229.9 3390.46
   283.1 3399.33   299.1 3404.87     307 3406.54   328.7 3408.82   339.8 3411.83
   371.6 3414.14   380.1 3416.06   392.1 3416.98   423.6  3423.3   452.6  3431.4
   483.5 3442.28   527.4 3452.46   599.4 3472.01   611.4 3474.29   638.5 3483.91
#Mann= 7 ,-1,0
       0      .1       0      30     .12       0     140      .1       0
   220.8    .045       0   229.9      .1       0  303.67     .12       0
  400.69      .1       0
Bank Sta=220.8,229.9
XS Rating Curve= 0 ,0
Exp/Cntr(USF)=0,0
Exp/Cntr=0.3,0.1

Type RM Length L Ch R = 1 ,13213   ,51.7,54.1,55
XS GIS Cut Line= 6
2319652.39338644659379.7439620712319581.11394754659226.625167403
2319515.11446708659176.4655622542319439.43506282659190.545451419
2319296.87618503659069.9864004452319165.75721718659070.866393517
#Sta/Elev= 30
       0 3453.97    73.4 3438.68    86.4 3434.59    95.5 3433.98   148.4 3417.93
   170.1 3407.01   175.1 3402.39   187.7 3387.78   190.2 3385.58   193.4 3384.81
   210.3 3388.52   219.1 3385.73   230.5  3385.7   250.6 3393.02   275.1 3397.68
   287.3 3397.82   295.5 3399.14   319.9 3405.86   343.3 3409.14   349.5 3408.69
   383.1 3411.96   401.1 3415.38   448.3 3426.94   505.2 3444.86   520.2 3447.57
   556.2 3458.62   568.2 3459.94   592.2 3465.27   628.2 3476.06   646.6  3480.4
#Mann= 7 ,-1,0
       0      .1       0      50     .12       0     130      .1       0
   219.1    .045       0   230.5      .1       0  338.77     .12       0
  368.77      .1       0
Bank Sta=219.1,230.5
XS Rating Curve= 0 ,0
Exp/Cntr(USF)=0,0
Exp/Cntr=0.3,0.1

Type RM Length L Ch R = 1 ,13159   ,32.8,32.9,33.8
XS GIS Cut Line= 6
2319683.11896528659353.6384321672319611.83952638659200.519637499
2319545.84004592659150.3600323492319470.16064166659164.439921514
2319327.60176387659043.8808705412319196.48279602659044.760863613
#Sta/Elev= 30
       0  3447.9     8.6 3446.51    25.9 3441.57    83.8 3430.03   132.9 3417.96
   159.1  3407.2   168.1 3402.32   182.5 3392.01   195.13380.085   198.6 3379.09
   202.4 3380.07   218.7 3380.97   242.4 3384.71   289.9 3397.69   298.2 3397.44
   326.7 3400.18   338.2 3402.49   355.2 3403.04   362.8 3406.12   375.1    3409
   420.5 3417.54   467.6 3431.21   502.8 3439.08   518.9 3445.28   558.9 3454.23
   582.9 3461.82   590.9 3462.53   602.9 3465.81   626.9 3468.82   646.6    3474
#Mann= 3 ,-1,0
       0      .1       0   195.1    .045       0   202.4      .1       0
#XS Ineff= 2 , 0
                          216.82         3385.21
Permanent Ineff=
       F       F
Bank Sta=195.1,202.4
XS Rating Curve= 0 ,0
Exp/Cntr(USF)=0,0
Exp/Cntr=0.3,0.1

Type RM Length L Ch R = 1 ,13126   ,71.6,70.8,71.4
XS GIS Cut Line= 6
2319705.94320033 659330.783088512319634.66376144659177.664293842
2319568.66428098659127.5046886922319492.98487671659141.584577857
2319350.42599892659021.0255268832319219.30703107659021.905519956
#Sta/Elev= 30
       0 3442.68    77.8 3424.39   153.1 3402.55   176.3 3390.13   182.1 3385.36
   192.1 3374.35   203.83371.618     211  3370.5   215.23371.468   239.5 3378.07
   252.3  3383.1   256.4 3386.18   268.6 3387.57   276.7 3391.39   288.9 3391.25
     297 3392.24   305.1 3394.74   329.8 3399.48   366.6 3402.17   387.5 3406.35
   426.1 3416.73     463 3425.21   502.8 3437.07   517.7 3442.68   549.6 3450.93
   565.7 3453.43   585.7 3458.06   613.2 3466.11   625.7 3466.64   646.6 3470.98
#Mann= 3 ,-1,0
       0      .1       0   203.8    .045       0   215.2      .1       0
Bank Sta=203.8,215.2
XS Rating Curve= 0 ,0
Exp/Cntr(USF)=0,0
Exp/Cntr=0.3,0.1

Type RM Length L Ch R = 1 ,13056   ,24.8,20.6,19.3
XS GIS Cut Line= 6
 2319758.7427847659281.5034764332319687.46334581659128.384681765
2319632.40721227659087.9057296662319552.93972638659096.513945368
2319403.22558329658971.7459148062319272.10661544658972.625907879
#Sta/Elev= 30
       0 3435.38    66.5 3418.04   119.8 3401.12   128.3 3399.73   154.8  3391.9
   167.8 3384.88   181.1 3373.73   187.8 3369.47   204.53361.988   207.7 3361.44
   216.5 3361.95   232.6 3364.25   276.7 3378.83   293.8 3382.02   328.6 3390.54
   366.1 3393.28   378.6 3395.14   406.7  3403.7   422.3 3409.63   453.6 3419.69
   466.1 3425.16   474.4 3430.35     482 3432.04   500.4 3439.26   519.1 3445.12
   543.1 3451.33   559.1 3453.53   583.1 3458.83   603.1 3465.49   643.2 3471.09
#Mann= 3 ,-1,0
       0      .1       0   204.5    .045       0   216.5      .1       0
Bank Sta=204.5,216.5
XS Rating Curve= 0 ,0
Exp/Cntr(USF)=0,0
Exp/Cntr=0.3,0.1

Type RM Length L Ch R = 1 ,13035   ,34.8,38.1,45.6
XS GIS Cut Line= 6
2319765.91782152 659266.076528612319684.40861686659084.728298152
2319619.88866948659083.1344568682319556.28058541659088.917009965
2319404.65543207658964.7928219162319283.35101572658963.213337328
#Sta/Elev= 30
       0 3432.76     9.8 3431.04    35.3 3422.98    62.4 3416.28   150.3  3388.5
   168.4 3381.01   185.2 3371.22   189.6 3369.31   198.3 3368.32   207.1 3362.17
   215.9 3360.01   219.1 3359.61   224.1 3359.96   255.1 3366.08   285.9 3378.25
   303.2 3380.73   323.3 3386.82   342.9 3390.59   377.3 3393.75   396.3 3397.66
   459.4 3419.53   472.1 3424.55   482.5 3430.66     491 3432.36   523.2 3444.11
   548.4 3451.33   586.5 3459.19   611.7 3468.16   631.7  3472.4   644.5 3473.62
#Mann= 3 ,-1,0
       0      .1       0   215.9    .045       0   224.1      .1       0
#XS Ineff= 2 , 0
          210.05 3366.03  232.26         3368.17
Permanent Ineff=
       F       F
Bank Sta=215.9,224.1
XS Rating Curve= 0 ,0
Exp/Cntr(USF)=0,0
Exp/Cntr=0.3,0.1

Type RM Length L Ch R = 1 ,12997   ,145.7,146.8,149
XS GIS Cut Line= 6
2319780.05607274659258.9777367912319695.08785271659071.636989292
2319640.03171918659031.1580371932319560.56423329659039.766252894
 2319410.8500902658914.9982223332319351.01056125658913.238236188
#Sta/Elev= 30
       0 3433.81     6.4  3432.1    19.5 3426.39    59.1  3416.8    76.6 3410.24
    92.3 3405.81     103  3401.2   142.5 3389.45   160.1 3383.07   194.7 3373.61
   212.4 3359.35   218.1 3356.13   223.9 3354.46   230.1 3354.37   242.7 3347.31
     249  3346.8     259 3347.39     286 3355.97   301.2 3364.35   322.2 3378.43
   330.2 3381.68   342.3 3385.74   370.1 3390.39   390.9  3395.2   414.3 3402.47
   452.7 3416.53     469 3424.46   498.1 3436.16   567.5  3458.6   608.7 3475.75
#Mann= 3 ,-1,0
       0      .1       0   242.7    .045       0     259      .1       0
Bank Sta=242.7,259
XS Rating Curve= 0 ,0
Exp/Cntr(USF)=0,0
Exp/Cntr=0.3,0.1

Type RM Length L Ch R = 1 ,12850   ,84.7,84.9,84.5
XS GIS Cut Line= 4
2319842.92004011659170.6466721222319800.15237677658984.607336601
 2319740.2776481658915.4662808712319458.72386445658864.145084865
#Sta/Elev= 30
       0 3411.68    34.3 3400.07    66.9 3384.62    91.8 3375.64   145.2 3349.69
   161.6 3346.83   173.9 3340.78   186.2  3337.5   190.3 3336.69     199 3337.93
   209.2  3337.5   218.8  3335.1   227.5 3334.17   238.7 3335.23   245.9 3337.12
     250 3339.28   269.5 3354.84   274.8 3357.95   290.6 3363.51   314.4 3366.91
   344.3 3367.46   371.9 3369.86   384.1 3372.05   394.5 3375.21   428.8 3388.94
     441 3392.03   449.5 3397.56   473.6 3408.22   518.3 3427.82   568.5 3448.03
#Mann= 3 ,-1,0
       0      .1       0   218.8    .045       0   238.7      .1       0
#XS Ineff= 2 , 0
          204.04 3342.16
Permanent Ineff=
       F       F
Bank Sta=218.8,238.7
XS Rating Curve= 0 ,0
Exp/Cntr(USF)=0,0
Exp/Cntr=0.3,0.1

Type RM Length L Ch R = 1 ,12765   ,339.2,341.8,339.8
XS GIS Cut Line= 4
2319886.25766754 659044.827687922319865.36346841658930.327476675
2319773.42899222 658828.363784912319615.46884678658806.633817812
#Sta/Elev= 30
       0 3358.19      20 3342.96    39.3 3331.14    44.4 3329.42    56.5 3327.91
    64.7  3327.9      81 3329.22    97.2 3328.57   128.7 3330.55   134.1 3329.46
   139.5 3326.85     148 3326.27   155.6 3325.44   160.5 3326.21   174.7 3333.72
   183.9 3342.52   198.7 3352.83   213.7 3358.28     259  3364.2   271.1 3368.67
   289.6 3369.11   299.4 3371.33   311.5 3372.71   319.5 3375.06   339.7 3376.38
   351.9 3379.83     364 3381.44   380.1 3385.33   392.2  3389.6   413.1 3398.83
#Mann= 3 ,-1,0
       0      .1       0     148    .045       0   160.5      .1       0
#XS Ineff= 2 , 0
           127.5 3339.41
Permanent Ineff=
       F       F
Bank Sta=148,160.5
XS Rating Curve= 0 ,0
Exp/Cntr(USF)=0,0
Exp/Cntr=0.3,0.1

Type RM Length L Ch R = 1 ,12423   ,163.4,168.5,172.4
XS GIS Cut Line= 4
 2320140.7033792658926.6137201512320109.52575262658787.873281898
2320048.20975369658695.8992835052319995.72741563658643.416945439
#Sta/Elev= 30
       0 3334.29     5.6 3332.32      22 3328.15    41.8 3325.92    58.6 3324.81
    71.2 3322.63    83.5 3319.11    98.7 3316.08   124.5 3313.07   132.7 3309.42
   145.4 3302.16   156.7  3301.8   164.7 3299.32     174 3295.01   180.7 3293.25
   194.2 3292.74   199.9 3291.76   207.9  3291.1   213.43291.669   222.4 3294.77
   238.4 3305.59   246.4 3312.93   252.7 3317.32   258.4 3322.21   264.1 3327.56
   268.8 3333.06   274.5  3338.6   291.5 3352.82   301.8 3357.35     327 3365.88
#Mann= 3 ,-1,0
       0      .1       0   199.9    .045       0   213.4      .1       0
Bank Sta=199.9,213.4
XS Rating Curve= 0 ,0
Exp/Cntr(USF)=0,0
Exp/Cntr=0.3,0.1

Type RM Length L Ch R = 1 ,12255   ,138,137.3,136.1
XS GIS Cut Line= 3
2320232.33494706658856.0713536362320240.69262671658690.589296509
2320193.88962066658625.399395216
#Sta/Elev= 30
       0 3317.44    18.9 3312.15    26.9 3311.13    30.9 3310.95    42.9 3308.81
      67    3307      71  3305.4    82.7 3298.21      91 3291.23      95 3288.89
     103 3287.14     115  3278.8     119 3277.29   127.1 3276.65   135.1 3277.06
   138.2 3278.15   143.1  3279.8   147.1 3280.74   155.1 3283.93   159.1 3285.93
   163.1 3287.28   169.9  3288.9   182.2 3291.22     192  3295.8   201.5 3299.18
   211.7 3306.57   218.7  3310.2   226.5 3315.06     233 3318.08   245.9 3327.05
#Mann= 3 ,-1,0
       0      .1       0     115    .045       0   138.2      .1       0
Bank Sta=115,138.2
XS Rating Curve= 0 ,0
Exp/Cntr(USF)=0,0
Exp/Cntr=0.3,0.1

Type RM Length L Ch R = 1 ,12118   ,270.4,259.9,256.5
XS GIS Cut Line= 4
2320348.72971124658864.4382407882320376.88948957658767.639002779
2320370.72953806658628.6000972762320348.80495065658592.782443228
#Sta/Elev= 30
       0 3313.46     7.6 3311.36    15.9 3310.93    20.1 3309.99    28.4    3307
    55.3 3287.48    61.7 3281.87    65.9 3278.97    78.4 3275.72    82.5 3275.26
    86.7 3275.39      95 3278.78      99 3278.43   111.3 3274.85   119.3 3270.73
     1223270.013   135.3 3269.43   141.8 3269.97   151.3 3271.35   159.3 3273.83
   167.3 3277.74   179.3 3285.62   183.4 3287.56   203.5 3299.61   211.2 3303.45
   218.9 3306.21   232.5 3308.77     256  3312.2   276.3 3316.47     282 3318.35
#Mann= 3 ,-1,0
       0      .1       0     122    .045       0   141.8      .1       0
Bank Sta=122,141.8
XS Rating Curve= 0 ,0
Exp/Cntr(USF)=0,0
Exp/Cntr=0.3,0.1

Type RM Length L Ch R = 1 ,11858   ,214.1,220,226.2
XS GIS Cut Line= 3
2320652.69580086658905.2535250962320641.72589521658841.743545038
2320487.56985271658671.421325792
#Sta/Elev= 30
       0 3291.16     7.4 3283.06    12.3 3278.57    16.3 3275.48    31.7 3269.06
    52.8 3257.82    66.8 3253.78    82.9    3252    93.6 3249.41    99.9 3249.03
   113.8  3249.4   119.2 3249.86     130  3251.8   144.3 3252.13   159.4 3254.66
   173.1 3259.81   178.5 3263.08   182.1 3263.67   191.9    3264   200.1 3266.77
   210.9 3269.38   227.4 3277.91   241.5 3286.35   248.6 3289.91     254 3291.64
   259.4 3292.55   264.2  3292.8     281 3297.33   286.4 3297.93   294.2 3297.73
#Mann= 3 ,-1,0
       0      .1       0    93.6    .045       0   113.8      .1       0
Bank Sta=93.6,113.8
XS Rating Curve= 0 ,0
Exp/Cntr(USF)=0,0
Exp/Cntr=0.3,0.1

Type RM Length L Ch R = 1 ,11638   ,135.1,138.6,143.4
XS GIS Cut Line= 4
2320705.80865034658776.2413082772320740.90830785658741.921643158
2320744.02827741658645.9825793032320732.71838777 658606.20296746
#Sta/Elev= 30
       0 3257.02     3.3 3256.49    10.1 3256.54    14.5 3256.91    23.6  3255.9
      35 3255.88    44.4 3254.77    48.1 3253.67    49.8 3252.86    57.8 3247.79
    64.6 3244.01    69.8 3240.58    73.8 3238.25    77.8 3236.97    89.9 3236.59
    93.9  3236.1   101.9 3234.68   105.9 3232.98   108.5 3232.67   109.9 3232.44
   124.73232.712   129.9 3233.15   133.9 3234.11   145.1 3241.93   148.8  3244.9
   162.5  3254.9   168.3  3258.8   179.2 3267.53   183.3 3269.64   186.4  3270.9
#Mann= 3 ,-1,0
       0      .1       0   108.5    .045       0   124.7      .1       0
Bank Sta=108.5,124.7
XS Rating Curve= 0 ,0
Exp/Cntr(USF)=0,0
Exp/Cntr=0.3,0.1

Type RM Length L Ch R = 1 ,11499   ,124.7,123.1,121.1
XS GIS Cut Line= 3
2320761.40882508658858.600340344 2320905.1723254 658662.29676562
2320886.11933138658596.477331742
#Sta/Elev= 30
       0  3264.7     6.7 3262.25    31.5 3256.39    57.4 3252.91    66.2 3250.13
    80.3 3248.72      91 3245.63   103.2 3244.28   106.2 3243.15   114.6 3236.02
   126.5 3227.61   134.6 3223.62   146.8 3221.38   153.6 3220.92   163.3 3220.92
   174.7 3222.49   183.3 3219.52   194.7  3218.7   196.33219.185   200.1  3220.9
     215 3231.62   229.8  3244.7   234.8 3248.55   239.7 3251.19   248.6 3253.89
     257 3255.17   269.5 3258.39   293.5 3265.22   302.8 3268.65   311.8 3270.52
#Mann= 3 ,-1,0
       0      .1       0   183.3    .045       0   196.3      .1       0
Bank Sta=183.3,196.3
XS Rating Curve= 0 ,0
Exp/Cntr(USF)=0,0
Exp/Cntr=0.3,0.1

Type RM Length L Ch R = 1 ,11376   ,301.8,307,311.3
XS GIS Cut Line= 4
2320910.36859649658874.766517086 2320962.9086709658811.256537028
2320992.93157057658724.0746553122320994.66366093658636.315410142
#Sta/Elev= 30
       0  3249.3    16.6 3241.35    21.7 3239.52    30.8 3237.49      45 3232.62
    59.2 3229.73    65.6 3227.19    71.9 3223.56    79.1 3216.25    84.6 3212.54
    88.2 3211.76    93.1 3211.78    97.3 3210.84   105.8 3206.55     110 3205.08
   118.5 3205.25   122.7 3204.65   126.9 3202.76   130.93201.792   135.4  3201.5
   142.3 3201.79   148.1  3202.8   160.8 3207.33   189.5  3225.4   205.5 3234.42
   221.5 3244.92   241.5 3252.45   249.5  3256.4   253.5 3257.79   262.4 3259.63
#Mann= 3 ,-1,0
       0      .1       0   130.9    .045       0   142.3      .1       0
#XS Ineff= 2 , 0
          117.49 3213.28
Permanent Ineff=
       F       F
Bank Sta=130.9,142.3
XS Rating Curve= 0 ,0
Exp/Cntr(USF)=0,0
Exp/Cntr=0.3,0.1

Type RM Length L Ch R = 1 ,11069   ,204.2,206.7,205.8
XS GIS Cut Line= 3
2321036.45635491659053.4522573172321233.96591126658951.764168904
2321358.14271153658819.765207982
#Sta/Elev= 30
       0 3263.85    13.2 3256.36    26.7 3246.63    32.7 3243.14    44.7 3232.76
    53.7 3227.43    63.6 3219.09    80.7  3206.2    86.1 3203.62    94.2 3198.34
    98.7 3196.66   103.2 3193.98   114.2 3186.01   116.7 3184.98   130.2 3182.45
   139.2 3177.55   141.83176.946   145.5 3176.62   159.23177.006   161.6 3177.29
   166.1 3179.68   179.6 3191.74   197.6 3203.03   206.6  3209.9   215.6 3214.06
   228.4  3215.9   282.1 3226.12     348 3239.52   358.5 3240.79   403.4 3252.17
#Mann= 3 ,-1,0
       0      .1       0   141.8    .045       0   159.2      .1       0
Bank Sta=141.8,159.2
XS Rating Curve= 0 ,0
Exp/Cntr(USF)=0,0
Exp/Cntr=0.3,0.1

Type RM Length L Ch R = 1 ,10862   ,175,175.9,176.1
XS GIS Cut Line= 2
2321109.78911098659205.9843899382321454.94194954659102.340761362
#Sta/Elev= 30
       0 3243.78     2.5 3243.31    10.8 3239.08    23.4 3230.34    40.1 3223.99
    58.4 3213.17    69.3 3209.35    81.8 3206.27    86.1 3203.35   102.7 3186.51
   106.9 3183.22   111.1 3181.37   119.4 3173.46   123.6 3171.32   140.3 3165.02
   152.8 3165.57   163.2 3164.07   169.5 3163.65   175.5 3164.06   182.1 3166.03
   190.4 3171.99   207.1 3174.91   219.7 3181.87   223.8 3183.15   253.1 3187.59
   262.7 3190.49   269.2  3192.9   301.3 3208.48   332.4 3221.41   360.4 3229.43
#Mann= 3 ,-1,0
       0      .1       0   163.2    .045       0   175.5      .1       0
Bank Sta=163.2,175.5
XS Rating Curve= 0 ,0
Exp/Cntr(USF)=0,0
Exp/Cntr=0.3,0.1

Type RM Length L Ch R = 1 ,10687   ,159.5,159.4,159.4
XS GIS Cut Line= 3
2321059.91346683 659329.805973322321253.87300148659338.542889295
2321479.28543364659293.110926224
#Sta/Elev= 30
       0 3251.89    16.3 3245.12    32.3 3235.76    44.3 3232.07    56.3 3227.02
    64.3 3221.37    68.3 3220.17    80.3 3214.13    92.4 3210.15    96.4 3207.68
   116.4  3190.7   120.4 3188.86   124.4 3185.72   132.4 3177.36   144.4  3167.7
   152.4 3162.71   164.4 3159.97   184.4 3158.78   204.7 3161.16   214.2 3161.08
   216.9 3160.76   225.1 3156.08   233.2 3154.23   236.13154.251   249.13154.856
   261.8 3159.56   278.8 3170.57   331.2 3193.49   367.9 3203.93   424.1 3226.25
#Mann= 3 ,-1,0
       0      .1       0   236.1    .045       0   249.1      .1       0
Bank Sta=236.1,249.1
XS Rating Curve= 0 ,0
Exp/Cntr(USF)=0,0
Exp/Cntr=0.3,0.1

Type RM Length L Ch R = 1 ,10527   ,164.6,168.5,170.6
XS GIS Cut Line= 3
2321085.34485896659473.8933921042321260.36570344659500.293184288
2321544.89679698659440.649209353
#Sta/Elev= 30
       0 3226.48     2.9 3225.25      19 3221.66    39.3 3210.36    51.4 3206.72
    67.6 3198.64    87.8 3192.51   104.3 3186.37   128.3 3181.18   142.5 3180.21
   156.5 3178.06   168.7 3177.61   176.8 3175.87   180.9 3174.38   193.4 3164.87
   209.5 3154.01   217.7 3151.16   225.8  3150.8   240.3 3145.99   246.3 3145.17
   253.8    3146   270.8 3154.03     279 3155.81   287.2 3158.76   307.6 3170.56
   323.9 3178.17   356.6 3190.98   405.8 3208.07     422 3212.81   467.7 3231.95
#Mann= 3 ,-1,0
       0      .1       0   240.3    .045       0   253.8      .1       0
Bank Sta=240.3,253.8
XS Rating Curve= 0 ,0
Exp/Cntr(USF)=0,0
Exp/Cntr=0.3,0.1

Type RM Length L Ch R = 1 ,10359   ,54,53.5,50.9
XS GIS Cut Line= 3
2321090.23370936659596.1146522162321419.74222663659669.447408284
2321550.76341747659656.736397232
#Sta/Elev= 30
       0 3209.43     6.1 3206.29    14.3  3204.2    30.7 3196.39    56.1 3186.87
    79.8 3179.65    99.7 3174.56   145.4 3157.78   165.9 3151.07   174.1 3146.78
   178.2  3146.1   186.4 3142.96   218.23133.184   223.7 3132.56   233.1  3133.2
   243.8 3136.03   260.2 3137.13   288.8 3140.46   309.3 3144.12   317.6 3144.18
   350.1 3149.57   370.2 3158.14   378.2 3160.49   402.3 3173.25   414.4 3177.49
   426.4  3183.2   434.5 3188.86   450.5 3196.57   466.6 3205.66   469.2  3207.7
#Mann= 3 ,-1,0
       0      .1       0   218.2    .045       0   233.1      .1       0
Bank Sta=218.2,233.1
XS Rating Curve= 0 ,0
Exp/Cntr(USF)=0,0
Exp/Cntr=0.3,0.1

Type RM Length L Ch R = 1 ,10305   ,40.6,35.6,33.9
XS GIS Cut Line= 4
2321089.30143338659651.2289976442321274.93962198659696.078560015
2321328.75909683659697.6385447932321545.59698099 659667.21884162
#Sta/Elev= 30
       0 3207.84       4 3205.45    15.3  3201.2    30.5  3193.8    53.7 3185.42
    89.4 3174.18   101.7 3165.76   109.9  3163.5   118.2 3159.46   146.5    3149
   159.8 3143.41   169.7  3140.8     184 3138.16   192.2 3134.91   196.2 3133.89
   204.2 3133.06   210.63131.495   216.6 3131.05   227.73131.546   244.2 3135.18
   260.4 3135.52   304.8 3141.37   316.9 3141.86   349.2  3148.1   356.4 3150.59
   369.4 3156.45   377.5 3159.11   401.8  3172.8   413.9 3176.15   463.8 3201.76
#Mann= 3 ,-1,0
       0      .1       0   210.6    .045       0   227.7      .1       0
Bank Sta=210.6,227.7
XS Rating Curve= 0 ,0
Exp/Cntr(USF)=0,0
Exp/Cntr=0.3,0.1

Type RM Length L Ch R = 1 ,10269   ,168.8,164.9,165.1
XS GIS Cut Line= 4
2321085.20334724659666.9983442062321256.48967588659752.290511951
2321381.09346003659694.7270736382321542.55188457659671.210303107
#Sta/Elev= 30
       0 3204.28    16.7 3197.66    30.1  3191.2      48 3185.64    75.4 3175.07
    85.7 3172.83    92.7 3170.05     115 3156.32   126.4 3153.41   141.8 3147.63
   159.7 3145.37   164.2  3143.8   186.5 3128.84   195.4 3125.67   208.6 3122.86
   217.6 3122.91   229.33121.088   239.5 3120.75   244.7 3121.09   262.8 3123.43
   268.8 3125.89   277.8 3131.56   284.6 3133.83   335.8 3141.31   347.9 3141.61
   384.3 3148.91   408.5 3158.54   432.8  3172.4     444 3175.47   491.8 3199.91
#Mann= 3 ,-1,0
       0      .1       0   229.3    .045       0   244.7      .1       0
#XS Ineff= 2 , 0
          218.77 3128.14
Permanent Ineff=
       F       F
Bank Sta=229.3,244.7
XS Rating Curve= 0 ,0
Exp/Cntr(USF)=0,0
Exp/Cntr=0.3,0.1

Type RM Length L Ch R = 1 ,10105   ,157.2,165.8,173.8
XS GIS Cut Line= 3
2321142.93471555659869.3284984052321361.90592246659887.715393642
 2321577.5340575659712.204120931
#Sta/Elev= 30
       0  3152.8     5.3 3151.04    21.3  3148.7    29.3 3148.92    45.4 3146.78
    82.5 3144.92    97.6 3141.64   133.7 3137.22   141.7 3135.09   150.5 3134.61
   173.8 3128.88   185.9 3128.49   197.9 3126.48   219.7 3118.52   238.1 3116.18
   248.5 3113.02   274.5 3114.14   288.6 3110.31   296.23109.611   306.1 3109.48
   312.1 3109.53   318.8  3110.4   337.8 3118.37   361.9 3133.39   375.8 3144.08
   390.9 3152.92   416.5 3172.11   464.8 3202.09   476.2 3207.95   497.8 3214.63
#Mann= 3 ,-1,0
       0      .1       0   296.2    .045       0   312.1      .1       0
Bank Sta=296.2,312.1
XS Rating Curve= 0 ,0
Exp/Cntr(USF)=0,0
Exp/Cntr=0.3,0.1

Type RM Length L Ch R = 1 ,9939    ,107.4,115.4,121.9
XS GIS Cut Line= 3
2321331.36982141 659932.540492932321552.01256425660029.489576903
2321581.26444304660023.639201146
#Sta/Elev= 30
       0 3121.03      14 3118.45    22.7 3114.55    35.8 3111.75    44.6  3108.9
    53.3 3107.47      62 3103.74    70.8 3104.09    75.2 3105.67    79.5 3106.18
    92.6 3106.13      97    3105   101.6 3103.05   110.1 3101.44     1193097.103
   127.6  3096.5   133.53097.094   143.8 3099.33   153.8 3105.46   162.5  3112.8
   179.6  3125.3   184.4 3129.67   193.1  3135.6   207.5 3147.09   210.8 3149.98
   223.7 3163.53     241 3178.06   257.5 3186.62   265.6 3188.83   270.8 3191.78
#Mann= 3 ,-1,0
       0      .1       0     119    .045       0   133.5      .1       0
Bank Sta=119,133.5
XS Rating Curve= 0 ,0
Exp/Cntr(USF)=0,0
Exp/Cntr=0.3,0.1

Type RM Length L Ch R = 1 ,9823    ,93.6,84.8,70.5
XS GIS Cut Line= 4
2321282.54557531659943.3909124172321356.26783176660014.676069481
2321371.49970293660079.8684780772321511.02364282660079.259203231
#Sta/Elev= 30
       0  3127.8    30.1 3121.48    36.4 3120.68    48.6 3117.27      59 3116.17
    63.5 3114.96    87.3 3105.05    96.9 3102.09   102.6 3098.53   114.5 3089.55
   119.7 3086.69   121.6 3085.69   133.9 3084.83   138.2  3086.2   146.2 3089.78
   150.3 3090.53   154.4 3090.93   194.2 3090.69   198.2 3091.19   206.2 3093.91
   210.2 3095.91   214.2 3098.92   226.2 3109.66   238.2 3118.51   247.8 3127.35
   270.2  3146.1   282.2 3154.79   294.2 3162.17   298.2 3164.01     309 3166.36
#Mann= 3 ,-1,0
       0      .1       0   119.7    .045       0   138.2      .1       0
Bank Sta=119.7,138.2
XS Rating Curve= 0 ,0
Exp/Cntr(USF)=0,0
Exp/Cntr=0.3,0.1

Type RM Length L Ch R = 1 ,9739    ,38.6,38.9,42.3
XS GIS Cut Line= 4
2321200.01665349660023.1764868082321254.57749999660095.404655037
2321415.14227685 660115.670112312321512.31254633660103.199061681
#Sta/Elev= 30
       0 3133.06     6.9 3130.52    15.8 3128.99    33.4 3124.16    78.6 3114.72
   104.2 3102.38     115 3095.39   124.4 3090.28   132.4 3086.74   140.5 3080.39
   144.5 3079.02   160.7 3077.12   168.8 3076.78   179.5 3077.22   184.9 3078.81
   190.2 3081.23     197 3082.82     205 3086.27     209 3086.78   217.1 3084.66
   229.6 3086.97   241.3 3091.41   249.4 3095.32   261.5 3103.39   273.8 3114.06
   289.7 3126.66   305.5 3140.78   317.9 3150.09     330 3157.76   350.3 3165.85
#Mann= 3 ,-1,0
       0      .1       0   160.7    .045       0   179.5      .1       0
Bank Sta=160.7,179.5
XS Rating Curve= 0 ,0
Exp/Cntr(USF)=0,0
Exp/Cntr=0.3,0.1

Type RM Length L Ch R = 1 ,9700    ,92.7,89.1,85.2
XS GIS Cut Line= 4
2321205.21292458660050.1970965052321262.89153374660125.023400282
2321370.45434542660158.7991624042321493.08634328 660127.62153583
#Sta/Elev= 30
       0 3127.75     4.2 3126.28    18.9 3122.48    34.1 3120.31    41.3 3118.24
    49.9 3116.52    59.3 3113.78    84.6 3109.56    95.8 3104.22     100 3101.36
   112.6  3091.4   129.4 3077.19   133.9 3074.82   143.5 3072.22   146.7 3071.68
   159.33072.091   162.9 3072.98   167.1 3075.84   178.6 3077.78   191.3 3080.72
   204.8 3080.14   217.2 3081.71   225.5 3086.93   233.8 3089.54   246.1 3095.39
   262.6 3107.68     275 3115.11   299.8 3135.36   316.3 3148.16   333.8 3155.33
#Mann= 3 ,-1,0
       0      .1       0   143.5    .045       0   159.3      .1       0
Bank Sta=143.5,159.3
XS Rating Curve= 0 ,0
Exp/Cntr(USF)=0,0
Exp/Cntr=0.3,0.1

Type RM Length L Ch R = 1 ,9611    ,185.5,181.9,183.7
XS GIS Cut Line= 4
2321192.74187395660191.0160431972321227.55689029660228.948822195
2321425.53481904660213.8796360182321474.89939445660171.270213034
#Sta/Elev= 30
       0 3113.29    22.8 3108.89    40.9 3103.02    56.1 3098.97    72.2 3087.34
    80.2 3080.15    96.2 3069.12     1023068.001   116.3 3067.26   121.33068.004
   132.3 3071.48   139.2 3072.16   160.4 3071.43   172.5 3073.72   176.5 3073.55
   184.5 3071.81   189.8 3071.65   196.5 3072.38   204.5 3074.84   212.6 3074.46
   216.6 3075.04   220.6 3076.56   236.6 3079.42   240.7 3080.91   251.1 3087.28
   264.1 3098.25   275.1 3105.02   289.3 3116.99   295.8 3123.82   315.2    3138
#Mann= 3 ,-1,0
       0      .1       0     102    .045       0   121.3      .1       0
Bank Sta=102,121.3
XS Rating Curve= 0 ,0
Exp/Cntr(USF)=0,0
Exp/Cntr=0.3,0.1

Type RM Length L Ch R = 1 ,9429    ,93,92,94
XS GIS Cut Line= 4
 2321217.1643481660285.5881771382321272.76444882660335.472379656
 2321429.1722088660359.3752266962321470.22275046660354.698582709
#Sta/Elev= 30
       0 3101.82    25.5 3097.09    57.8 3089.48    63.2 3087.65    73.9 3085.46
    78.1 3083.54    86.2 3077.09    94.3 3071.57   106.5 3065.03   110.5 3063.86
   122.7 3064.82   126.7 3063.39   146.9 3053.49     151 3054.03   159.1 3056.42
   167.2  3057.4   171.2 3057.34   175.3 3056.57   189.83051.493   191.4 3050.79
   195.5 3050.48   203.6 3051.51   207.6 3052.42   211.7 3055.44   227.9 3069.02
   235.9 3076.39   244.8 3083.29   256.1 3091.03   268.2 3102.08   274.2 3105.69
#Mann= 3 ,-1,0
       0      .1       0   189.8    .045       0   203.6      .1       0
#XS Ineff= 2 , 0
          168.95  3060.3
Permanent Ineff=
       F       F
Bank Sta=189.8,203.6
XS Rating Curve= 0 ,0
Exp/Cntr(USF)=0,0
Exp/Cntr=0.3,0.1

Type RM Length L Ch R = 1 ,9337    ,81.1,82.2,80.9
XS GIS Cut Line= 3
2321243.61418506660395.5559457012321391.54511492660451.552399375
2321443.36272876660434.837040069
#Sta/Elev= 30
       0 3082.62     9.2 3079.27    26.3 3075.86    34.8 3072.93    43.4 3070.98
    47.6 3068.93    56.2 3062.19    60.5 3059.43    64.8 3057.79    76.2 3056.62
    82.4 3057.46    86.1  3057.3    90.4 3055.21    94.8 3051.65      99 3047.68
   103.2 3044.95   107.5 3044.43   119.6 3044.41     132 3044.58   135.8 3045.31
   141.7 3047.21   144.4 3049.03   158.2 3060.84   167.2 3066.75   176.4 3071.89
   184.1 3077.02   195.5 3083.22     205 3088.86   208.2 3090.46   212.6 3092.11
#Mann= 3 ,-1,0
       0      .1       0   103.2    .045       0   135.8      .1       0
Bank Sta=103.2,135.8
XS Rating Curve= 0 ,0
Exp/Cntr(USF)=0,0
Exp/Cntr=0.3,0.1

Type RM Length L Ch R = 1 ,9255    ,19.6,19.6,18.8
XS GIS Cut Line= 4
2321203.65404325660467.4576654852321290.95139766660501.233427606
2321368.89546409660526.6951559752321449.95729319660473.693190799
#Sta/Elev= 30
       0 3088.84     7.9 3086.17    17.7 3081.59    30.6  3077.5    56.3  3066.9
    69.2 3055.33    73.5  3051.9    77.8 3049.34      82 3048.27    99.1 3046.79
   103.3 3044.58   107.5 3041.28   115.9 3036.53   120.1 3035.84   124.3 3035.83
     137 3036.22   148.5 3036.92     158 3038.87   166.4 3038.72   170.7 3039.07
     193 3046.57   210.9 3055.46   217.8 3059.47   222.5 3062.97   229.5 3066.63
   236.8 3070.24   251.2 3075.91   258.8 3079.34   265.5 3083.32   272.5 3086.63
#Mann= 3 ,-1,0
       0      .1       0   115.9    .045       0     137      .1       0
Bank Sta=115.9,137
XS Rating Curve= 0 ,0
Exp/Cntr(USF)=0,0
Exp/Cntr=0.3,0.1

Type RM Length L Ch R = 1 ,9235    ,47.7,46.7,43.9
XS GIS Cut Line= 4
 2321202.2372071660499.2398771312321281.41997606660522.934285902
2321359.32219605660534.9188160122321444.52843549660481.619181043
#Sta/Elev= 30
       0 3083.76    10.4 3081.56    22.9 3075.89    31.2 3072.55    48.1 3061.24
    56.3 3055.37    64.7 3048.63    68.8 3046.06      73 3045.09    81.4 3044.19
    85.4 3043.34    89.5  3041.7   101.6 3035.37   107.43034.004   113.8 3033.69
   121.5 3034.01   138.1 3034.87   142.1 3035.54   146.1 3037.04   150.2 3038.06
   162.5 3037.62   167.2 3038.58   189.5  3045.7   195.3 3047.85   200.2 3050.23
   209.7 3055.31   221.4 3062.74   232.6 3068.54   247.4 3075.02     262 3082.23
#Mann= 3 ,-1,0
       0      .1       0   107.4    .045       0   121.5      .1       0
Bank Sta=107.4,121.5
XS Rating Curve= 0 ,0
Exp/Cntr(USF)=0,0
Exp/Cntr=0.3,0.1

Type RM Length L Ch R = 1 ,9188    ,70.6,66.1,62.7
XS GIS Cut Line= 4
2321193.26150106660579.1774940412321256.24661876660575.209455639
2321368.89546409660565.6671891922321444.76102209660512.145596907
#Sta/Elev= 30
       0 3082.65     5.3 3080.48      23  3070.9      43 3057.99      51 3049.19
      55 3045.63      59 3042.72    63.1 3040.28    67.1  3039.2    71.1 3038.75
    75.1 3037.45    79.1 3035.74    83.1 3033.15    87.1 3029.09    91.1 3024.35
    95.2 3020.63   106.53019.322   119.2    3019   124.1 3019.36   139.3 3023.44
   153.7 3030.03   171.4 3035.76   199.8 3041.71   207.6  3042.5   211.7 3043.41
   227.7 3050.57   244.9 3061.71   253.6 3068.11   263.4  3070.6     269 3072.58
#Mann= 3 ,-1,0
       0      .1       0   106.5    .045       0   124.1      .1       0
Bank Sta=106.5,124.1
XS Rating Curve= 0 ,0
Exp/Cntr(USF)=0,0
Exp/Cntr=0.3,0.1

Type RM Length L Ch R = 1 ,9122    ,144,139.5,137
XS GIS Cut Line= 3
2321201.82578679660649.6294071492321298.77487077660645.450567322
2321425.81160149660591.961417544
#Sta/Elev= 30
       0 3078.31     6.4 3075.81    22.4 3067.62    34.4 3062.71    54.4 3051.04
    58.4 3048.29    62.4 3044.52    66.4    3039    70.4 3034.39    74.4 3032.91
    82.4 3032.51    86.4 3031.01    90.4 3028.82   102.9 3020.31     108 3017.52
   111.6 3016.62   124.6 3015.42   133.3 3015.89   137.53017.532   146.3  3022.2
   153.3 3024.43   159.3 3025.12     168 3024.29   171.6 3024.63   189.9 3029.62
   202.7 3032.18   207.1 3034.38   215.7 3039.96   220.5 3042.07   234.9 3051.22
#Mann= 3 ,-1,0
       0      .1       0     108    .045       0   137.5      .1       0
Bank Sta=108,137.5
XS Rating Curve= 0 ,0
Exp/Cntr(USF)=0,0
Exp/Cntr=0.3,0.1
